HEC-RAS study ARNOLDCK.prj: ARNOLDCK

--- ARNOLDCK.g01 (geometry) --- (continued)

Type RM Length L Ch R = 1 ,43468.7 ,199.5,199.5,199.6
XS GIS Cut Line= 2
     1596375.764      287660.612     1597119.002      288074.301
#Sta/Elev= 30
       0  870.56    48.9  850.33      88  835.85   117.3  821.92   127.1  818.08
   136.9  815.06   156.4  810.29   185.8  804.54   215.1  801.59   234.6  801.87
     264  803.65   283.5  803.66     352  802.15   449.8  798.53   518.2  796.89
   557.3  794.83   567.1  793.84   587.4  790.15   596.4  789.87   602.4  791.71
   606.2  792.88   625.7  802.92   674.6  823.27   713.7  837.88   733.3  842.61
   743.1  847.17   762.6  868.02   772.4  874.93   821.3  898.01   850.6  912.72
#Mann= 3 , 0 , 0
       0     .06       0   587.4    .045       0   602.4     .08       0
#XS Ineff= 2 , 0
           266.2   804.1
Permanent Ineff=
       F       F
Bank Sta=587.4,602.4
XS Rating Curve= 0 ,0
Exp/Cntr=0.3,0.1

Type RM Length L Ch R = 1 ,43269.2 ,1482.9,1443.1,1407.8
XS GIS Cut Line= 4
     1596269.643      287676.884     1596383.366      287884.261
     1596818.191      288131.777     1597025.569      288145.156
#Sta/Elev= 30
       0  861.86    37.8     849    47.3  846.74    75.7  842.04   170.3  815.57
   179.8  813.58   189.2  812.52   236.5  809.83     266  806.34   285.6  804.62
   334.6  803.76   393.5  804.26   422.9  803.72   619.1  795.58   648.6  793.23
   668.2  790.06     678   789.8   687.1  791.36     727   800.7   746.3  806.31
   765.2  813.24   821.9  835.93   831.3  838.82   850.2  842.54   859.6  845.92
   869.1  851.14   897.4  869.12   906.9  874.39   916.3  878.72   944.7  890.06
#Mann= 3 , 0 , 0
       0     .06       0   668.2    .045       0   687.1      .1       0
#XS Ineff= 2 , 0
          392.96  804.63
Permanent Ineff=
       F       F
Bank Sta=668.2,687.1
XS Rating Curve= 0 ,0
Exp/Cntr=0.3,0.1

Type RM Length L Ch R = 1 ,41826   ,665,670.7,671.9
XS GIS Cut Line= 4
     1595865.729      288895.175     1596475.814      288853.798
      1596548.72      288675.179     1597004.276      288258.513
#Sta/Elev= 30
       0 1019.44    67.9 1006.68   135.9  996.92   203.8  983.47   252.4  971.91
   281.5  961.92   407.7  911.93   475.6  890.82   524.1  877.23   611.5  859.32
   698.3  808.16     708  804.43   717.6  802.18   775.5  790.75   785.1  789.03
   794.2  788.96   804.4  790.52     824     794   833.8  794.75   961.2  799.43
  1059.2   799.4  1196.4  796.08  1235.6  797.22  1245.4  800.22  1255.2  805.05
    1314  836.04  1323.8  839.34  1343.4  843.69  1382.6  868.01  1421.8  886.94
#Mann= 3 , 0 , 0
       0     .06       0   775.5    .045       0   804.4     .06       0
#XS Ineff= 2 , 0
                          966.76          801.24
Permanent Ineff=
       F       F
Bank Sta=775.5,804.4
XS Rating Curve= 0 ,0
Exp/Cntr=0.3,0.1

Type RM Length L Ch R = 1 ,41155.3 ,1048.4,1075.3,1101.9
XS GIS Cut Line= 3
     1596934.831      289111.291     1597093.165      288905.735
     1597379.276      288491.846
#Sta/Elev= 30
       0  849.35     9.6  844.42    28.8  835.43    38.4  831.46    57.7  825.44
    67.3  822.92    86.5  818.93   144.2  808.95   153.8  807.94   192.2  805.69
   259.5  801.01   375.6  793.94   404.6  792.58     424   792.5   433.6  791.72
     453  788.42   462.7  788.04   472.3  789.02   520.7  797.63   569.1  806.81
   578.8  809.39   588.4  812.57   627.2  826.38   636.8  828.49   646.5  829.98
   656.2   832.5   665.9  836.48   704.6   854.4   743.3  872.96   762.6   882.9
#Mann= 3 , 0 , 0
       0     .06       0     453    .045       0   472.3     .08       0
Bank Sta=453,472.3
XS Rating Curve= 0 ,0
Exp/Cntr=0.3,0.1

Type RM Length L Ch R = 1 ,40080   ,774.7,783.1,791.4
XS GIS Cut Line= 2
     1596339.572      289331.019     1598537.302      289944.675
#Sta/Elev= 30
       0  998.78    98.4  991.07   383.6   981.2   422.9  977.29   472.1  960.05
   501.6  946.44   678.6  846.65     777  798.77   796.7  794.68   855.7   790.3
   865.5  786.95   875.3  786.72   885.2  788.15   914.7     794     954  795.57
  1170.4  789.59  1190.1  791.58  1258.9  825.84  1288.4  834.19  1426.1  909.73
  1583.5  975.99  1603.2  981.86  1701.5  997.24  1740.8 1007.43  1760.5 1008.11
    1908  995.75  1976.9  985.53  2035.9  983.09  2153.9  985.76  2281.8  993.75
#Mann= 3 , 0 , 0
       0     .06       0   855.7    .045       0   885.2     .06       0
Bank Sta=855.7,885.2
XS Rating Curve= 0 ,0
Exp/Cntr=0.3,0.1

Type RM Length L Ch R = 1 ,39297   ,829.5,807.8,786.1
XS GIS Cut Line= 3
     1596676.498      289639.068     1596815.387      290047.402
      1597248.72      290364.068
#Sta/Elev= 30
       0  909.24    58.8  881.42    78.4   871.8   117.6  851.96   137.2   842.8
     147  838.74   156.8  835.12   225.5  811.15   235.3  808.51   245.1  807.09
   254.9  806.33   284.3  804.48   303.9  803.54   528.9  797.32     607  793.28
   665.5  791.09   714.3  788.39   724.1  787.24   733.8  786.77   743.6  786.85
   753.3  788.05   782.6  796.88   792.4  800.02   802.1  803.46   821.6  811.22
   850.9  824.26   860.7  827.72   880.2   831.6     890  835.47     968  878.54
#Mann= 3 , 0 , 0
       0     .06       0   714.3    .045       0   753.3      .1       0
Bank Sta=714.3,753.3
XS Rating Curve= 0 ,0
Exp/Cntr=0.3,0.1

Type RM Length L Ch R = 1 ,38489.1 ,1051.6,1059.5,1066.5
XS GIS Cut Line= 2
     1595815.506      291110.204     1597105.127      290717.828
#Sta/Elev= 30
       0  972.59    19.7  966.44    49.2     954      59  954.36   137.8   987.8
   157.4  994.34   177.1  998.85   255.8 1006.78   285.3 1006.66   314.9 1003.15
   393.6  980.89   442.8  961.48   521.5  920.84   659.2  846.59   708.4  826.46
     738  816.47   787.2  811.74   806.8  808.44     856  789.61   865.9   787.1
   880.9  785.43   895.4   785.1   895.9  785.19   924.9  790.89  1052.8   791.8
  1249.6  797.85  1259.4  800.34  1308.6  821.53  1338.2  828.53    1348  832.68
#Mann= 3 , 0 , 0
       0      .1       0   880.9    .045       0   895.9     .06       0
Bank Sta=880.9,895.9
XS Rating Curve= 0 ,0
Exp/Cntr=0.3,0.1

Type RM Length L Ch R = 1 ,37429.6 ,974.7,1000.1,1026.5
XS GIS Cut Line= 3
     1596833.631       291482.43     1597102.572      291541.597
     1597783.162      291544.247
#Sta/Elev= 30
       0   904.9    29.5  892.06    78.7  874.06   108.2  864.11   137.7  852.54
     177  839.89     236  822.15   275.4  809.62   285.1  807.54   294.8  806.36
   421.2  798.02   567.1  789.27   576.8  788.25   603.6  782.89   615.7  782.42
   618.6  782.78   644.8  787.38     674  794.33   693.4   800.8   712.9  809.19
   722.6  812.55   742.1  817.18   751.8  822.07   761.5  828.26   810.1  862.63
   819.8  868.79   858.7  887.53   887.9  903.24   917.1  921.04     956  947.22
#Mann= 3 , 0 , 0
       0      .1       0   603.6    .045       0   618.6      .1       0
Bank Sta=603.6,618.6
XS Rating Curve= 0 ,0
Exp/Cntr=0.3,0.1

Type RM Length L Ch R = 1 ,36429.5 ,397.9,395.7,393.6
XS GIS Cut Line= 2
     1596495.822      291565.741     1597106.933      293044.908
#Sta/Elev= 30
       0    1005   117.8   995.3   137.5  991.32   157.1  983.41   206.2  959.05
   314.2   900.2   333.8  886.28   363.3  859.16   382.9  843.34   441.8  804.48
   461.5  789.09   471.3  783.43   481.1  780.92   500.8  780.33   549.8  785.38
   589.1  787.34   628.4  787.88   638.2  787.09     648  783.96   667.7  781.05
   677.5  783.07   697.1  791.06   716.8   793.8    1031  794.16  1296.1  810.62
  1315.7  814.81  1364.8  833.32  1413.9  843.74  1472.8  862.12  1600.4  896.08
#Mann= 3 , 0 , 0
       0     .06       0     648    .045       0   677.5     .06       0
Bank Sta=648,677.5
XS Rating Curve= 0 ,0
Exp/Cntr=0.3,0.1

Type RM Length L Ch R = 1 ,36033.7 ,804.1,819.6,835.1
XS GIS Cut Line= 2
     1596235.118      292028.121     1596765.866      292997.254
#Sta/Elev= 30
       0  857.63    48.9  841.29    97.8   823.2   117.3  814.73   156.4   795.5
   166.2  791.55     176  788.35   185.8  785.99   195.6  784.74   224.9     785
   273.8  783.13   293.3  781.66   308.3  780.92   312.9   780.9   322.7  781.92
   342.2  785.61   361.8  787.72   469.4  793.65   498.7  794.18   625.8  794.01
   762.7  794.47   831.2  796.31     880  799.09   997.4  811.52  1007.2  813.13
  1016.9  815.67  1026.7  818.83  1065.8  832.71  1075.6   835.1    1105  839.96
#Mann= 3 , 0 , 0
       0     .06       0   293.3    .045       0   308.3     .06       0
Bank Sta=293.3,308.3
XS Rating Curve= 0 ,0
Exp/Cntr=0.3,0.1

Type RM Length L Ch R = 1 ,35214.1 ,798.7,796.8,794.8
XS GIS Cut Line= 2
     1595902.233      291920.272     1595707.472      292989.845
#Sta/Elev= 30
       0  882.67    58.8  873.69   146.9  864.98   176.3  861.36   205.7  856.89
   235.1  849.65   264.4  844.39   274.2  841.34   323.2  820.37   352.6  811.25
   362.4  806.36     382  793.44   391.8  788.54   401.6  786.55   695.4  785.14
   734.6  784.37   754.2  782.25     764  781.03   773.7  780.99   783.3   782.1
   822.7  792.78   861.9   802.2   891.3   810.9   940.2  824.05     950  827.82
   959.8  833.16   969.6  839.36    1048  889.98  1067.6  901.88  1087.2  912.81
#Mann= 3 , 0 , 0
       0     .06       0   754.2    .045       0   783.3     .06       0
Bank Sta=754.2,783.3
XS Rating Curve= 0 ,0
Exp/Cntr=0.3,0.1

Type RM Length L Ch R = 1 ,34417.3 ,802.2,782.3,761.5
XS GIS Cut Line= 3
     1595381.594       291887.19      1595287.15      292626.079
     1595464.928      292909.413
#Sta/Elev= 30
       0  863.11      49  852.13    88.2  841.89     196  804.73   225.4  793.39
     245  784.98   254.8  781.54   262.7  780.94   264.6   780.8   277.7   780.8
   323.4  780.93   372.4  783.92   421.5  786.12   499.9   788.2   627.3  790.58
   744.9  795.17   784.2  796.17   813.8  796.03   823.6  796.69   833.4  798.53
   882.6  812.71   902.3   817.7     922  821.38   951.5   824.8   961.3  827.51
     981  836.61   990.8   840.6  1010.5  847.13    1040   855.2  1079.4  864.97
#Mann= 3 , 0 , 0
       0      .1       0   262.7    .045       0   277.7     .06       0
Bank Sta=262.7,277.7
XS Rating Curve= 0 ,0
Exp/Cntr=0.3,0.1

Type RM Length L Ch R = 1 ,33635   ,502.5,511.4,522.8
XS GIS Cut Line= 5
     1593570.483      291548.302     1594519.079      291987.465
     1594551.377      292152.547     1595170.483      292792.746
     1595492.705      292953.857
#Sta/Elev= 30
       0  924.16     127  947.47   234.5  949.84   420.1  943.55   459.2  940.33
   498.2  941.56   605.7  954.23   713.2  954.99   722.9  952.56   771.8  929.66
   830.4  909.19   918.3  861.97   937.9  854.11    1016  855.95  1045.3  851.85
  1157.5  801.36  1185.5     794    1256  781.35  1272.2  780.41    1282  780.89
  1370.1  785.96  1448.4  786.87  1888.8  783.88    2016  791.94  2035.6  795.76
  2084.6  812.85  2104.1   816.8  2191.8  816.96  2289.1  824.89  2464.4   877.6
#Mann= 3 , 0 , 0
       0      .1       0    1256    .045       0    1282     .06       0
Bank Sta=1256,1282
XS Rating Curve= 0 ,0
Exp/Cntr=0.3,0.1

Type RM Length L Ch R = 1 ,33123.6 ,90.9,82.9,72.8
XS GIS Cut Line= 3
     1592518.248      291455.055     1594669.712      292706.251
     1594975.702      292737.501
#Sta/Elev= 30
       0  825.98    19.7  828.38    78.7  827.42   236.1  840.81   334.5  842.04
     423  839.38   452.5  833.77   501.7  817.54   531.2  810.84   570.6  794.69
   590.2  789.85   629.6  794.09     846  801.48  1249.3  799.55  1446.1  806.53
    1574  815.31  1800.2  817.14    1938  805.45  2006.8   794.3  2085.5  791.68
  2124.8  794.32  2213.4  791.13  2262.6  787.09    2292  779.51    2307   779.2
    2361  780.39  2410.1  792.19  2449.5  791.96  2508.1   787.1  2796.4  787.61
#Mann= 3 , 0 , 0
       0     .06       0    2292    .045       0    2307     .06       0
#XS Ineff= 2 , 0
                         2421.13          792.59
Permanent Ineff=
       F       F
Bank Sta=2292,2307
XS Rating Curve= 0 ,0
Exp/Cntr=0.3,0.1

Type RM Length L Ch R = 1 ,33040.7 ,69.9,60.5,49.4
XS GIS Cut Line= 3
     1594309.144       292553.06     1594673.728      292760.004
     1594764.006       292778.06
#Sta/Elev= 30
       0  801.82   126.7  796.54   175.5  794.99   185.2  794.28     195  793.17
   204.7  791.68   214.5  789.12   224.2  786.05     234  783.43   253.5  781.29
     273  779.51   282.7  779.56   292.5  781.89   302.2  783.52   321.7  784.87
   331.5  785.08     351  783.92   370.5  784.58   380.2  785.23     390   787.1
   399.7  790.96   409.5  795.81   419.2  800.01   428.4  801.39   437.6  801.81
     456  802.23   474.5  802.38   483.7  802.01   502.1  800.95   511.3  800.78
#Mann= 3 , 0 , 0
       0     .06       0   253.5    .045       0   282.7     .06       0
Bank Sta=253.5,282.7
XS Rating Curve= 0 ,0
Exp/Cntr=0.3,0.1

Type RM Length L Ch R = 1 ,32980.2 ,82.4,86.5,89.6
XS GIS Cut Line= 5
     1594390.394      292686.393     1594564.006      292741.949
     1594680.672      292775.282     1594811.228      292798.893
     1595184.004      292820.196
#Sta/Elev= 30
       0  813.13      48  810.77    86.3   811.9    95.9  811.25   115.1  808.65
   134.3  807.76   143.9  804.81   153.5  798.82   172.7  783.54   182.3  779.83
   191.6  778.79     201  778.61   219.6  778.91   238.3  780.44   247.6  782.07
     257   785.1   266.3  790.21   275.6  796.82     285  802.53   294.3  806.17
   303.6  808.02   341.5  808.44     370  806.46   398.4  806.22   436.3  808.43
   485.4  809.94   573.8  814.09   603.3  814.93   652.5   815.8   809.7  815.89
#Mann= 3 , 0 , 0
       0     .06       0   182.3    .045       0   238.3     .06       0
Bank Sta=182.3,238.3
XS Rating Curve= 0 ,0
Exp/Cntr=0.3,0.1

Type RM Length L Ch R = 1 ,32893.7 ,317.9,311.3,307.7
XS GIS Cut Line= 5
     1594375.117      292748.893     1594548.728      292804.449
     1594712.617      292848.893     1595014.006      292871.115
     1595571.156      293073.668
#Sta/Elev= 30
       0   819.9    57.6  812.96   124.7  813.63   153.5  811.75   163.1  808.48
   201.2  785.66   210.6   781.9     220  779.66   229.4  778.72   267.2  778.38
   276.6  778.48   304.9  779.82   333.2  783.67   352.1  784.49   469.1  794.22
   488.6  794.88   566.6  795.52   751.5  790.79     839  790.35   877.8  787.47
     907  788.69   926.4  792.79   936.1  796.31   965.3  809.68   984.7  816.04
   994.4  820.23  1023.6  836.56    1043  844.44  1188.8  895.07  1247.1  913.18
#Mann= 3 , 0 , 0
       0      .1       0     220    .045       0   276.6      .1       0
#XS Ineff= 2 , 0
                          557.01          795.61
Permanent Ineff=
       F       F
Bank Sta=220,276.6
XS Rating Curve= 0 ,0
Exp/Cntr=0.3,0.1

Type RM Length L Ch R = 1 ,32582.4 ,746.3,756.4,766.5
XS GIS Cut Line= 3
     1594278.936      293106.185     1594667.825      293085.352
     1595535.881      293328.407
#Sta/Elev= 30
       0  970.02    19.5  962.26    58.4  944.38    97.4  924.72   126.6  911.02
     185  881.27   214.2  867.37   350.5  807.55     370  799.73     409  786.28
   428.6  780.35   438.4  778.26   442.1  777.94   448.2   777.4     458   777.4
   487.4  777.64     507  778.39     703  787.41   830.4  788.84   957.8   795.2
   967.5  796.37   977.3  799.44   996.9  808.59  1026.3  823.72  1104.7   865.3
  1124.3  874.98  1163.5  893.35  1222.3  918.68  1271.3  936.25  1290.9  944.08
#Mann= 3 , 0 , 0
       0      .1       0   442.1    .045       0     458     .06       0
Bank Sta=442.1,458
XS Rating Curve= 0 ,0
Exp/Cntr=0.3,0.1

Type RM Length L Ch R = 1 ,31826   ,676.5,683.3,690.1
XS GIS Cut Line= 3
     1594282.408       293599.24     1594594.908      293752.018
     1595049.498      294161.146
#Sta/Elev= 30
       0  868.65     9.7  866.43      29   863.5    67.6  858.76    77.3  856.46
   135.3  834.74   154.6  829.01   193.2  820.36   260.9  809.34   280.2  804.77
   318.9  793.58   338.2  788.89   357.6  782.74     377  780.53   425.5  781.53
   464.3  775.84   481.9  775.25   483.8  775.23   496.9  775.58   503.2  776.13
   512.9   778.5     542  789.25   648.8  835.62   784.7  888.96   813.8  902.49
   842.9  917.52   891.5  940.48   920.6  957.23     940  965.57   959.4  971.72
#Mann= 3 , 0 , 0
       0      .1       0   481.9    .045       0   496.9      .1       0
Bank Sta=481.9,496.9
XS Rating Curve= 0 ,0
Exp/Cntr=0.3,0.1

Type RM Length L Ch R = 1 ,31142.6 ,764.6,749.4,734.2
XS GIS Cut Line= 2
     1593950.683      293696.991     1594443.738      294519.908
#Sta/Elev= 30
       0  978.38    48.9  950.21   107.7  917.73   127.3  907.72   195.8  880.35
   254.5  860.42   274.1  852.77   293.7  846.48   352.4  829.51   362.2   825.7
   450.3  782.42   460.1   777.9   469.9   774.8   479.7  773.85   489.4  773.83
   489.6  773.84   499.2  774.24     509  775.56   538.4  780.95     558  783.58
   606.9  786.71   636.3  787.76   685.2  787.04   734.2  787.49     744  789.75
   753.8  793.78   832.1  829.84   900.6  859.13     930  870.16   959.3  878.34
#Mann= 3 , 0 , 0
       0      .1       0   469.9    .045       0   489.6      .1       0
Bank Sta=469.9,489.6
XS Rating Curve= 0 ,0
Exp/Cntr=0.3,0.1

Type RM Length L Ch R = 1 ,30393.2 ,790.9,778.1,765.1
XS GIS Cut Line= 2
     1593085.045      294438.598     1594084.209      294814.497
#Sta/Elev= 30
       0 1089.86    19.6 1083.54    29.4 1082.43      49 1083.52    68.6 1081.36
    97.9 1073.58   117.5 1065.81   205.7 1025.94   225.3 1015.92   254.6  997.34
   323.2  949.93   342.8  939.15     382  920.95   528.9  855.44   587.6  830.16
     617  816.47   646.4  800.99     666   792.1   695.4  782.39     715  777.65
   734.5  774.77   754.1  773.38   765.2  773.66   780.2  774.55   842.3  778.94
   861.9  781.23   969.6  805.47     999  811.27  1018.6  813.42  1067.5  815.05
#Mann= 3 , 0 , 0
       0      .1       0   765.2    .045       0   780.2      .1       0
Bank Sta=765.2,780.2
XS Rating Curve= 0 ,0
Exp/Cntr=0.3,0.1

Type RM Length L Ch R = 1 ,29615.1 ,468.3,466.7,465
XS GIS Cut Line= 2
     1593335.511      295489.411     1593984.382      295357.032
#Sta/Elev= 30
       0  911.87      39  886.29    58.4  872.77    87.6  852.83    97.4  845.94
   107.1  838.86   116.9  832.01   126.6  825.58   165.6  801.65     185  789.14
   194.8  783.69   204.5  779.78   214.2  777.29     224  775.78   233.7  775.03
   253.2  774.15     263  773.49   272.7  773.06   282.4     773   311.6  773.14
   321.4  773.57   370.1  777.56   389.6  778.91     409  779.52     448  780.06
   467.5  780.87   486.9  782.03   516.2  784.37   574.6  789.58   662.2  799.73
#Mann= 3 , 0 , 0
       0      .1       0     263    .045       0   282.4      .1       0
Bank Sta=263,282.4
XS Rating Curve= 0 ,0
Exp/Cntr=0.3,0.1

Type RM Length L Ch R = 1 ,29148.4 ,497.9,508.5,519.1
XS GIS Cut Line= 3
     1593562.964      295794.379     1593691.436      295856.879
     1594222.686      295711.046
#Sta/Elev= 30
       0  834.24      19  830.56    57.2  825.64    66.7  823.97    76.2  821.53
   104.8  811.63   142.9   791.6   152.7  786.74   162.5  782.61   172.4   779.6
   182.2  777.63   211.7  773.54     219  773.07   231.4  772.78   241.2  772.85
   260.9  774.26   310.1  781.02   339.6  783.91   369.1  785.06     438  785.58
   477.4  788.42   516.7  792.91   536.4  796.19   595.4  811.85   624.9  818.68
   634.8  819.67   644.6  819.68   674.1  817.55   683.9  817.79   693.8  819.26
#Mann= 3 , 0 , 0
       0      .1       0     219    .045       0   241.2     .06       0
Bank Sta=219,241.2
XS Rating Curve= 0 ,0
Exp/Cntr=0.3,0.1

Type RM Length L Ch R = 1 ,28639.9 ,666,669.6,673.1
XS GIS Cut Line= 3
     1593404.955      296119.908     1593646.101      296214.526
     1594939.212      296471.932
#Sta/Elev= 30
       0     838    19.2  829.11    38.4  824.42    57.6  823.34   134.3  822.62
   153.5  820.34   201.5  808.36     259  789.94   278.7  785.25   347.6  781.85
   426.3  781.81   465.7  780.71   583.7   771.1   593.6  771.09   623.1  772.29
   701.8   781.1     751  782.97   760.8  785.84   790.4  801.69   859.2  831.89
  1065.9  912.91  1095.4  919.68    1184  934.43  1233.2  943.66  1262.7  947.18
  1311.9   948.1  1321.7  947.38  1351.2   942.4  1410.3  940.75  1577.5  929.65
#Mann= 3 , 0 , 0
       0      .1       0   583.7    .045       0   623.1      .1       0
#XS Ineff= 2 , 0
          424.76  781.85
Permanent Ineff=
       F       F
Bank Sta=583.7,623.1
XS Rating Curve= 0 ,0
Exp/Cntr=0.3,0.1

Type RM Length L Ch R = 1 ,27970.4 ,407,386.6,366.1
XS GIS Cut Line= 3
     1593284.016      296610.186     1593468.044      296783.797
     1594051.377      297006.019
#Sta/Elev= 30
       0  840.62    77.8  823.12   126.5  810.73     146  807.61   175.2  805.18
   184.9  803.95   204.3  799.88   214.1  796.32   223.8  791.82   243.3  781.06
     253  776.66   262.8  774.35   467.6   774.2   496.8  773.29   535.8  771.01
   565.1   770.5   574.9   770.5   604.1   770.5   613.9   772.5   623.6   777.2
   643.1  788.25   662.6  798.59   711.4  822.16   740.7  835.12   769.9  847.26
   799.2  858.42   818.7  865.09   838.2  871.12   857.7  876.09   877.2  878.78
#Mann= 3 , 0 , 0
       0     .06       0   574.9    .045       0   604.1      .1       0
Bank Sta=574.9,604.1
XS Rating Curve= 0 ,0
Exp/Cntr=0.3,0.1

Type RM Length L Ch R = 1 ,27583.8 ,836,825.8,815.7
XS GIS Cut Line= 2
     1593024.197       297404.68     1594191.732      297022.735
#Sta/Elev= 30
       0  931.22    68.8  901.72   157.2  865.91   304.6  803.97   353.8  783.54
   363.6  779.84   373.4  777.14   383.3  775.63   393.1  774.94   432.4  773.04
   471.7  771.64     511  770.66   540.5   770.5   560.2   770.5   589.6   770.5
     629  770.67   648.6  771.97   746.9  782.58   766.5  785.36   786.2  789.07
   815.7  795.59   835.3  800.51   874.6  811.89   933.6  827.72  1041.7   854.8
  1110.5   872.7  1169.5  886.08  1198.9  894.16  1208.8  897.19  1228.4  903.94
#Mann= 3 , 0 , 0
       0      .1       0   560.2    .045       0   589.6      .1       0
Bank Sta=560.2,589.6
XS Rating Curve= 0 ,0
Exp/Cntr=0.3,0.1

Type RM Length L Ch R = 1 ,26757.9 ,785.8,807.7,829.5
XS GIS Cut Line= 2
     1593866.211       298038.36     1594336.099      297349.075
#Sta/Elev= 30
       0  915.34    19.6  913.28     108  909.71   117.8  908.71   127.6  907.07
   147.2  902.57   255.2  870.04   284.6  861.76   333.7  848.81   343.5  845.83
   353.3  842.14   363.1  837.73   471.1  787.77   480.9   783.5   490.7  780.17
   500.5  777.97   510.3  776.37   539.8  772.36   556.8  770.65   569.2  770.13
   571.8  770.14   598.7  770.89   628.1  772.65   647.7  774.94   657.6  776.73
   667.4  780.05   677.2  785.25   696.8  797.61   706.6  802.58   834.2  861.13
#Mann= 3 , 0 , 0
       0      .1       0   556.8    .045       0   571.8      .1       0
Bank Sta=556.8,571.8
XS Rating Curve= 0 ,0
Exp/Cntr=0.3,0.1

Type RM Length L Ch R = 1 ,25950.3 ,275.2,279.8,284.5
XS GIS Cut Line= 2
     1594165.961      298164.352     1595129.232      298151.207
#Sta/Elev= 30
       0  839.59      59  828.93    88.5  823.99   137.6  816.55   206.4  806.94
   285.1   794.5   353.9     782   363.7  781.04   393.2  779.78   442.4  776.39
     462  773.98   501.3  767.65   516.1  766.87     521   766.8   531.1  766.84
   540.7  767.58   550.5  770.53   560.3  775.72   589.8  793.43   619.3   810.6
   658.6  835.04     698  860.38   756.9   899.7   786.4  919.08   815.9  937.46
   825.7  943.17   835.6  948.52   865.1  963.81   933.9 1000.52   963.4 1017.57
#Mann= 3 , 0 , 0
       0      .1       0   516.1    .045       0   531.1      .1       0
Bank Sta=516.1,531.1
XS Rating Curve= 0 ,0
Exp/Cntr=0.3,0.1

Type RM Length L Ch R = 1 ,25670.4 ,1075.3,1106.5,1137.7
XS GIS Cut Line= 2
     1594290.674      298351.038     1595461.679      298601.033
#Sta/Elev= 30
       0  804.52    39.3  799.58   166.8  780.05   176.7  779.35   186.5   779.3
   284.6  781.19   304.3  780.79   314.1  779.04   343.5  769.85   353.3  767.34
   363.1  766.19   368.1  766.19   383.1  766.49   392.6  767.07   402.4  769.18
   412.2   773.5   461.3   799.9   510.4   829.2   559.4  857.02   579.1  869.62
   628.1   903.3     687   942.2   736.1  972.21   745.9  977.81   755.7  982.23
   765.6  984.36   775.4  984.66     795  984.35   883.3  981.79  1197.4  970.75
#Mann= 3 , 0 , 0
       0      .1       0   368.1    .045       0   383.1      .1       0
Bank Sta=368.1,383.1
XS Rating Curve= 0 ,0
Exp/Cntr=0.3,0.1

Type RM Length L Ch R = 1 ,24564   ,835.1,853.8,872.4
XS GIS Cut Line= 2
     1593879.232      298376.902     1593918.294      299882.978
#Sta/Elev= 30
       0  812.29    97.8  791.64   127.2  787.19   156.5   784.5   244.6  780.63
   371.8   778.1   420.7   778.5   469.6  782.04   518.5  783.25   655.5  779.98
     675  778.43   753.3  763.76   772.9  761.82   776.2  761.87   791.2  762.39
     812  765.72   860.9  781.74   880.5  788.92   929.4  810.12  1017.4  867.31
  1115.3  924.14  1154.4  948.48  1213.1  987.88  1242.4  1005.4  1271.8 1021.45
  1340.3 1051.24  1477.2  1118.8    1487 1121.02  1496.8 1119.65  1506.6 1116.46
#Mann= 3 , 0 , 0
       0      .1       0   776.2    .045       0   791.2      .1       0
#XS Ineff= 2 , 0
          519.71  783.51
Permanent Ineff=
       F       F
Bank Sta=776.2,791.2
XS Rating Curve= 0 ,0
Exp/Cntr=0.3,0.1

Type RM Length L Ch R = 1 ,23710.2 ,1060,1039.4,1017.9
XS GIS Cut Line= 4
     1593492.349      298153.936     1593488.877      298456.019
     1593252.766      298667.825     1593159.016      298890.047
#Sta/Elev= 30
       0  900.55    19.5  890.62    29.2  885.05    68.2  860.45    87.7  850.95
   146.2  825.72   165.7   818.7   204.6  806.42   282.6  784.35   302.1  779.64
   330.9  774.38   359.8  772.68   398.2  771.46   494.3  771.75     504  771.02
   513.6  769.36   542.4  762.77     552  761.54   561.6  761.32     577  761.47
   590.5   761.8   600.1  763.58   609.7  767.93   648.2  789.77   667.5  801.22
   725.4  837.42   744.7  848.44     764  857.71   812.2   878.6   860.5  897.29
#Mann= 3 , 0 , 0
       0      .1       0     577    .045       0   600.1      .1       0
Bank Sta=577,600.1
XS Rating Curve= 0 ,0
Exp/Cntr=0.3,0.1

Type RM Length L Ch R = 1 ,22670.8 ,652.4,638.8,625.1
XS GIS Cut Line= 2
     1592374.891      297571.346     1592464.572      298733.797
#Sta/Elev= 30
       0 1056.34   186.2 1000.87   205.8  994.11   244.9  977.66   303.7  951.26
   372.3   916.6   411.5  895.88   431.1  886.49   480.1  867.64   538.9  848.26
   636.8  810.32   656.4  801.78   685.8  785.07   715.2  770.81   734.8  763.49
   744.6   760.7   754.4  759.16   764.2  758.83     774  758.96   803.4  760.01
   842.6  765.82   881.8  769.75   911.2  771.29   989.6     773  1009.1  774.86
  1077.7  792.68  1116.9  804.27  1126.7  807.61  1156.1  820.37  1165.9  823.47
#Mann= 3 , 0 , 0
       0      .1       0   754.4    .045       0     774      .1       0
Bank Sta=754.4,774
XS Rating Curve= 0 ,0
Exp/Cntr=0.3,0.1

Type RM Length L Ch R = 1 ,22032   ,307.6,299,290.5
XS GIS Cut Line= 2
      1591175.39      297608.014     1591960.045      298602.487
#Sta/Elev= 30
       0  892.02   127.7  902.29   166.9  910.01   255.3  931.12   304.4  937.95
     324  939.12   363.3   938.4   412.4   932.2   461.5  932.67   500.8  931.11
   520.4  924.46   569.6  896.57   608.8   868.8   648.1  838.48   667.8  825.45
   716.8  802.85   785.6  773.62   805.2  769.39   854.3  766.25   883.8  762.68
  1018.4  757.31  1021.3   757.3  1033.4   757.3  1050.7  757.72  1070.4  761.12
  1080.2  764.68  1109.6  780.08  1119.5  782.81  1227.5  792.83  1266.8  792.82
#Mann= 3 , 0 , 0
       0      .1       0  1018.4    .045       0  1033.4      .1       0
Bank Sta=1018.4,1033.4
XS Rating Curve= 0 ,0
Exp/Cntr=0.3,0.1

Type RM Length L Ch R = 1 ,21732.9 ,392.7,374.4,356.2
XS GIS Cut Line= 4
     1591396.297       298530.49     1591542.131      298527.018
     1591781.714       298655.49     1592035.186      298662.435
#Sta/Elev= 30
       0  870.76    19.4  858.18    68.1  828.56    77.8  821.96    87.5  814.12
     107  795.85   126.4  778.98   136.2  770.79   145.9  763.79   155.6  758.86
   165.5  755.86     175   754.8   180.5  754.72   194.4  754.65   204.1     755
   213.8  756.92     243  764.52   252.7   766.1   262.4  766.63   398.3  765.82
   417.7  766.55   437.2  770.03   476.2  779.55   505.5  785.11     525  787.96
   534.8  788.88   554.3  789.81   622.5  789.83     642  790.47   671.3  790.61
#Mann= 3 , 0 , 0
       0      .1       0   165.5    .045       0   180.5      .1       0
#XS Ineff= 2 , 0
                          260.28          767.38
Permanent Ineff=
       F       F
Bank Sta=165.5,180.5
XS Rating Curve= 0 ,0
Exp/Cntr=0.3,0.1

Type RM Length L Ch R = 1 ,21358.5 ,991.5,951.8,912.1
XS GIS Cut Line= 4
     1591070.268      300365.627       1591439.7      298956.387
     1591806.019      298849.935     1591951.853      298846.463
#Sta/Elev= 30
       0  870.16    39.1  889.92   166.2  931.02   244.4   947.7   303.1  953.32
   430.2   924.4   606.2  872.74   684.4  859.75   801.8  813.44   850.6  841.09
   889.8  842.69  1007.1  827.76  1046.2  813.24    1056  812.46  1095.1   827.7
  1124.4  832.26  1290.6   814.5  1329.8   804.6  1349.3  809.55  1398.2   833.4
  1417.8  836.49  1456.9   832.7  1593.8  760.64  1613.4  755.24  1623.1  754.69
  1642.7  755.25  1711.2  763.64    1809  765.72    1887  781.84  1984.2  789.16
#Mann= 3 , 0 , 0
       0      .1       0  1613.4    .045       0  1642.7      .1       0
Bank Sta=1613.4,1642.7
XS Rating Curve= 0 ,0
Exp/Cntr=0.3,0.1

Type RM Length L Ch R = 1 ,20406.7 ,795.7,834.3,873
XS GIS Cut Line= 4
     1592156.714      299867.296     1592076.853       299749.24
     1591917.131      299422.852     1591919.673      298886.245
#Sta/Elev= 30
       0  838.34    28.5  820.16    47.5  808.46      76  791.18   104.5  773.13
     114  768.36   123.5  764.89   142.5  758.41   152.4   755.2   162.2  753.35
     172  753.14   230.9  752.93   250.6  753.18   272.6  753.86     339  755.11
     388  756.54   574.2  762.94   593.7  763.75   603.5  764.42   613.2  765.68
     623  767.58   632.7   769.9   671.8  780.12   681.5  782.15   691.3  783.12
     701  783.36   749.8   783.9   779.1  784.79   847.4  786.37  1042.5  787.25
#Mann= 3 , 0 , 0
       0      .1       0   230.9    .045       0   272.6      .1       0
Bank Sta=230.9,272.6
XS Rating Curve= 0 ,0
Exp/Cntr=0.3,0.1

Type RM Length L Ch R = 1 ,19572.4 ,339,349.4,359.8
XS GIS Cut Line= 5
     1592330.325      299724.935     1592396.297      299551.324
     1592795.603      299384.657      1592936.75      299367.854
       1592974.7      298796.346
#Sta/Elev= 30
       0  842.26    29.3  832.73    48.9  824.06   185.7  771.01   205.4  764.85
   225.1  760.54   264.4  757.65   480.7  758.53   500.4  756.89   520.1  751.87
     535  750.61   539.7   750.6     550  750.78   559.4  752.43   579.1  758.99
   608.6  766.37   627.9  773.91   646.8   786.5   684.8  819.65   722.6  848.89
   741.6  861.84   760.6  872.78   847.9  875.69   935.3  884.99  1100.3  912.87
  1207.1  923.24  1226.5   919.5    1246  912.82  1275.1  901.71  1333.3  876.93
#Mann= 3 , 0 , 0
       0      .1       0     535    .045       0     550      .1       0
Bank Sta=535,550
XS Rating Curve= 0 ,0
Exp/Cntr=0.3,0.1

Type RM Length L Ch R = 1 ,19223   ,399.1,400.5,402
XS GIS Cut Line= 3
     1592341.413      299762.009     1592458.601      299735.967
     1592966.413      299768.519
#Sta/Elev= 30
       0  838.81    27.7  824.32    46.2  814.31     120   771.5   129.8  766.04
   139.6  762.84   149.4  762.18   266.8  759.02   276.6  758.52   286.4  756.82
     306  751.15   315.8  750.62   325.6   750.6   343.1   750.6   358.1   750.6
   384.3   750.6     394  750.85   403.8  752.51   413.6  757.49   423.4   765.1
   433.2  773.26   452.8  789.75   462.5  798.05   501.7  831.17     531  855.72
   540.8  863.64   550.6  870.54   560.4  876.32   589.8  892.35   628.9   913.9
#Mann= 3 , 0 , 0
       0     .08       0   343.1    .045       0   358.1      .1       0
Bank Sta=343.1,358.1
XS Rating Curve= 0 ,0
Exp/Cntr=0.3,0.1

Type RM Length L Ch R = 1 ,18822.5 ,650.7,628.2,605.8
XS GIS Cut Line= 3
       1592291.5       300033.71     1592488.983      300118.346
     1592792.802      300157.408
#Sta/Elev= 30
       0  850.47     9.8  847.09    29.3  839.87    39.1  835.94    68.4  823.71
    87.9  815.25    97.7  810.84   117.2  801.75     166  778.82   185.6   769.3
   195.3   765.3   205.1   762.8   214.8  760.61   224.4  757.12     234  752.93
   243.6  750.85   253.1  750.61   262.7   750.6   275.9   750.6   290.9   750.6
   329.7  750.66   339.3  751.31   348.9     753     368  757.31   377.6  759.61
   387.2   762.2   396.7  765.63   406.3  770.15   463.7  800.82   521.2  830.79
#Mann= 3 , 0 , 0
       0     .08       0   275.9    .045       0   290.9      .1       0
Bank Sta=275.9,290.9
XS Rating Curve= 0 ,0
Exp/Cntr=0.3,0.1

Type RM Length L Ch R = 1 ,18194.2 ,558.4,543,527.7
XS GIS Cut Line= 2
     1592297.634      301063.534     1592936.523      300323.951
#Sta/Elev= 30
       0  999.13    29.3  981.59    48.9  970.52   117.3  934.43   156.4  912.74
   195.5  892.13   205.2  886.84   224.8  875.77   244.3  864.04   263.9  851.61
     303   825.9   400.7  761.08   410.5  754.92   420.2   751.4   422.5  751.21
     430   750.6   439.8   750.6   488.7  750.64   498.4  750.94   576.6  755.85
   664.6  760.48   674.4  761.43   684.1  762.93   693.9  765.22   742.8  778.07
   772.1  785.47   801.4  792.49   869.8  808.11   928.5  820.23   977.3  830.89
#Mann= 3 , 0 , 0
       0      .1       0   422.5    .045       0   439.8      .1       0
Bank Sta=422.5,439.8
XS Rating Curve= 0 ,0
Exp/Cntr=0.3,0.1

Type RM Length L Ch R = 1 ,17651.2 ,919.3,932.2,945.1
XS GIS Cut Line= 2
     1593083.601      301239.005     1593116.153       300370.95
#Sta/Elev= 30
       0  987.08    29.3  973.27    48.8  963.02    68.3  952.12    87.8  940.26
   117.1  921.42   146.4  903.04     205  864.78   224.5  851.37   263.5  823.08
     283   809.6   302.6  796.68   312.3  791.25   341.6  776.65   351.4  772.37
   361.1  768.99   390.4   759.1   409.9  753.18   419.7  751.21   429.4  750.65
   439.2   750.6   452.8  750.74   478.2   752.1   614.9  762.73   634.4  764.98
   663.7  769.46     693   775.1   741.8     786   780.8  795.26   868.7  817.02
#Mann= 3 , 0 , 0
       0      .1       0   429.4    .045       0   452.8      .1       0
Bank Sta=429.4,452.8
XS Rating Curve= 0 ,0
Exp/Cntr=0.3,0.1

Type RM Length L Ch R = 1 ,16719   ,512.2,529.3,546.4
XS GIS Cut Line= 2
     1593722.686      301110.352     1594146.297      300492.296
#Sta/Elev= 30
       0  845.89    77.8  817.98   126.5  801.91     146  796.43   214.1   779.5
   272.5  764.16   282.2  762.23   301.7  760.51     360  756.83   408.7  754.32
   447.6  753.03   497.6  749.81     506   749.7   512.6  750.11   535.2   752.4
   544.9  754.05   554.7   756.6   564.4  759.61   574.1  763.18   583.9  767.27
   593.6  772.09   603.3  777.53   613.1  783.73   622.8  790.52   632.5  797.86
     652  813.83   690.9  848.03   710.4  864.53   729.8  879.83   749.3  894.01
#Mann= 3 , 0 , 0
       0     .08       0   497.6    .045       0   512.6      .1       0
Bank Sta=497.6,512.6
XS Rating Curve= 0 ,0
Exp/Cntr=0.3,0.1

Type RM Length L Ch R = 1 ,16189.7 ,458.6,463.7,468.7
XS GIS Cut Line= 2
     1593428.862      301348.164     1595189.979      300958.677
#Sta/Elev= 30
       0  950.93    29.4   939.8      49  933.27   274.5  867.82   372.5  837.18
   411.7  826.83   480.3  811.76   519.5  802.02     647  762.29   666.6  759.25
     745  753.24     794  744.92   794.3  744.93   803.8  745.14   809.3  746.66
   813.6  747.85   872.4  774.28   931.2  803.95   980.3  831.13  1107.7  903.99
  1205.7  957.95  1372.4 1052.79  1401.8 1067.95  1421.4 1076.06  1597.8 1142.84
  1666.4 1166.24  1744.9 1183.57  1764.5 1187.23  1784.1 1188.15  1803.7 1186.91
#Mann= 3 , 0 , 0
       0     .08       0   794.3    .045       0   809.3      .1       0
Bank Sta=794.3,809.3
XS Rating Curve= 0 ,0
Exp/Cntr=0.3,0.1

Type RM Length L Ch R = 1 ,15726   ,740.3,752.3,764.4
XS GIS Cut Line= 2
      1593696.94      301632.978     1594533.746      301636.451
#Sta/Elev= 30
       0  850.72    19.5  846.46    48.6  839.88    87.6  830.83     253  791.53
   272.4  787.26   301.6  781.14   340.6   773.3   379.5  765.15   389.2  763.42
     399  762.03   418.4  759.64   467.1  753.95   486.5  750.95     506  747.51
   515.7  745.58     523  744.45   525.4  744.08   535.2   744.1     538  745.06
   544.9  747.41   554.6  753.82   564.4  760.58   574.1  766.56   651.9  812.34
   729.8   857.8   739.5  863.26   749.2  868.41   778.4  883.27   836.8  912.65
#Mann= 3 , 0 , 0
       0     .08       0     523    .045       0     538      .1       0
Bank Sta=523,538
XS Rating Curve= 0 ,0
Exp/Cntr=0.3,0.1

Type RM Length L Ch R = 1 ,14973.7 ,1227.3,1234.1,1240.8
XS GIS Cut Line= 3
     1593580.771      301986.184     1593846.622      302253.111
     1594235.118       302485.76
#Sta/Elev= 30
       0  818.08      58  804.99   144.9  784.85   173.9  778.44   183.5  776.68
   202.9  773.86   251.2  767.79   280.1  763.64   309.1   758.5   328.4  754.01
   338.1  751.99   347.8  750.94   367.1  750.19   444.2  749.28   473.1  748.61
   482.7  747.93   492.4   746.9   521.2   743.2   530.9  742.12   540.5  741.74
   550.2  742.67   559.8   746.4   569.4  752.39   579.1  757.62     685  811.02
   704.3  820.28   752.5  842.36   781.4  855.95   810.3  870.11   829.6  880.14
#Mann= 3 , 0 , 0
       0     .06       0   521.2    .045       0   550.2      .1       0
Bank Sta=521.2,550.2
XS Rating Curve= 0 ,0
Exp/Cntr=0.3,0.1

Type RM Length L Ch R = 1 ,13739.6 ,743.1,759.5,775.6
XS GIS Cut Line= 3
     1592906.714      302891.602     1593319.908      303353.407
     1593385.881      303610.352
#Sta/Elev= 30
       0  852.63    78.7  815.58    88.5  810.56    98.4  804.96   147.5  773.41
   157.4  767.98   167.2  763.28   186.9  754.53   214.1  741.51   216.4  740.49
   226.2  739.24   236.1  740.43   255.7  744.64   265.6  745.27   373.8  743.06
   403.3   743.1   432.8     744   462.3   746.1   511.5  750.59   570.5  756.86
   649.2  763.02   668.8  765.58   688.4  769.58   698.3  772.31   717.9  779.53
   727.8  783.69   747.4  792.76   796.5  817.15   806.4  821.67     885  852.25
#Mann= 3 , 0 , 0
       0      .1       0   214.1    .045       0   236.1     .06       0
Bank Sta=214.1,236.1
XS Rating Curve= 0 ,0
Exp/Cntr=0.3,0.1

Type RM Length L Ch R = 1 ,12980.1 ,773.1,771.4,769.4
XS GIS Cut Line= 2
     1592481.604      303115.597     1592482.681      303841.219
#Sta/Elev= 30
       0  829.56   137.3  763.32   147.1  759.01   156.9  755.25   176.5  748.94
   186.3  746.77   196.1  745.46   215.7  744.45   294.2  744.05   323.6  744.86
   343.2   744.7   362.8   743.1   372.6  741.37   382.4  739.05   392.2  737.59
     402   738.3   421.6  743.96   431.4   745.1   460.9  745.32   470.7  746.35
   519.7  756.02   529.5  758.97   539.3  763.72   549.1  769.79   598.2  801.56
   686.4  861.43   696.2  867.72     706  872.97   715.8  876.95   725.6  880.47
#Mann= 3 , 0 , 0
       0      .1       0   382.4    .045       0     402      .1       0
Bank Sta=382.4,402
XS Rating Curve= 0 ,0
Exp/Cntr=0.3,0.1

Type RM Length L Ch R = 1 ,12208.8 ,424.5,404.3,384.3
XS GIS Cut Line= 4
     1588008.656      300248.321     1591743.519      303117.296
     1591802.547      303620.768     1591892.825      303731.879
#Sta/Elev= 30
       0  808.59      59  822.42   275.3  787.05   471.9  783.74   668.6   808.1
  1140.5   915.4  1494.5  773.15  1632.1  808.12  1966.4  763.08  2310.6  761.54
  2684.2  817.18  2821.8  828.69  2890.6  815.98  2998.8  854.53  3097.1  867.03
  3441.2  873.61  3814.9  845.68    3923  825.36    4100  763.32  4434.3  822.55
  4552.3  798.46  4758.3  826.47  4807.1  809.58  4885.1  751.24  4987.6  737.64
    5002   736.9  5011.8  737.46  5138.5  747.06    5226  792.64  5359.7  807.96
#Mann= 3 , 0 , 0
       0      .1       0  4987.6    .045       0  5011.8     .06       0
Bank Sta=4987.6,5011.8
XS Rating Curve= 0 ,0
Exp/Cntr=0.3,0.1

Type RM Length L Ch R = 1 ,11804.4 ,597.1,578.4,559.6
XS GIS Cut Line= 4
     1587897.545      301637.209     1591212.269      303412.435
     1591580.325      303700.629     1591802.547      303745.768
#Sta/Elev= 30
       0   933.5   147.3  994.15   274.9 1021.79   520.3 1022.46   598.9 1007.45
   981.8  802.58  1060.3  772.48    1129  793.02  1433.4  929.37  1521.7  952.81
  1600.3  938.72  1747.5  871.97  1875.2  852.66  1953.7  815.56  1973.4  817.62
  2169.7   915.5  2297.3  927.41  2503.5  904.64  2768.6  768.22  2964.9  861.02
  3269.3  883.54  3603.1  833.06    3662  813.48  3779.6  751.51    4004  737.08
  4013.4  736.12  4032.8  737.98  4217.9  750.93  4293.8   788.6  4454.4  801.41
#Mann= 3 , 0 , 0
       0     .06       0    4004    .045       0  4032.8     .06       0
Bank Sta=4004,4032.8
XS Rating Curve= 0 ,0
Exp/Cntr=0.3,0.1

Type RM Length L Ch R = 1 ,11226   ,279.2,273.4,267.4
XS GIS Cut Line= 3
     1590965.742      304058.268     1591625.464      303933.268
     1591851.158       303967.99
#Sta/Elev= 30
       0  903.68    29.2   881.8    68.1  849.26   165.4  778.06   194.6  757.73
   204.4  753.91   243.3  751.31     253  749.42   282.2  738.49   291.9  736.11
   301.7  735.86   321.1  740.52   330.9  743.17   340.6  743.96   408.7  746.77
   447.6  746.39   496.3  743.52   525.5  743.96   564.4  745.97     652  753.16
   661.7  754.81   671.5  758.24     700  773.24     719  785.92   728.6  790.27
   738.1  792.82   757.1  796.44   852.2  809.98   871.3  811.83   899.8  812.57
#Mann= 3 , 0 , 0
       0      .1       0   282.2    .045       0   321.1     .06       0
Bank Sta=282.2,321.1
XS Rating Curve= 0 ,0
Exp/Cntr=0.3,0.1

Type RM Length L Ch R = 1 ,10952.6 ,196.7,196.2,195.7
XS GIS Cut Line= 2
     1591130.545      304366.145     1591801.379      304045.312
#Sta/Elev= 30
       0  865.65    19.6  855.52    29.4  849.66    39.1  842.67    78.3  811.87
     137  764.03   146.8  756.94   156.6  752.54   166.3  751.17   185.9  751.01
   195.7  750.34   205.5  748.28   215.2  745.56   234.8   739.2   244.6  736.63
   254.4  735.87   264.2  737.02     274  739.42   283.7  741.66   293.5  742.59
   342.4  744.94   371.8  745.97   440.3     747   547.9  747.54   567.5   748.1
   577.3  749.34   587.1  751.96   665.3  779.25   684.9  784.08   743.6  796.85
#Mann= 3 , 0 , 0
       0      .1       0   234.8    .045       0     274     .06       0
Bank Sta=234.8,274
XS Rating Curve= 0 ,0
Exp/Cntr=0.3,0.1

Type RM Length L Ch R = 1 ,10756.4 ,51.2,51.2,51.2
XS GIS Cut Line= 2
      1591169.66      304572.382     1591828.515      304239.049
#Sta/Elev= 30
       0  785.65    19.4  782.58    48.6  781.05      68  781.69    97.2   785.1
   106.9  785.48     136  783.98   145.7   781.2   155.4  775.83   174.9  761.03
   184.6  755.04   194.3  751.73     204  751.13   233.2  751.51   252.6  749.94
     272  745.49   301.2  735.54   310.9  734.22   321.8   735.8     340  742.58
   359.5  746.47   369.2  747.38   456.6  744.09   534.4  744.16   563.5  745.25
   641.2  750.98   650.9   752.4   660.6  755.15   699.5  771.84   738.4  785.76
#Mann= 3 , 0 , 0
       0     .06       0   301.2    .045       0   321.8     .06       0
Bank Sta=301.2,321.8
XS Rating Curve= 0 ,0
Exp/Cntr=0.3,0.1

Type RM Length L Ch R = 1 ,10705.3 ,207.7,208.4,209.3
XS GIS Cut Line= 2
     1591197.265      304615.611     1591856.119      304282.278
#Sta/Elev= 30
       0  771.38    29.2  765.73    58.3  758.18    77.7  754.48   106.9  751.85
     136  750.98   155.4  749.69   174.9  747.46   194.3  747.49   213.7  748.55
   223.5  748.15   262.3  743.08     272  741.23   301.2  734.01   310.9  733.75
   320.4   734.7     340  741.44   349.8  744.04   369.2   747.4   378.9  747.44
   398.3  744.49   437.2  741.69   495.5  741.91   524.6  742.89   573.2   745.7
   641.2   751.6   650.9  753.35   670.4  759.86     719  781.44   738.4  789.34
#Mann= 3 , 0 , 0
       0     .06       0   301.2    .045       0   320.4     .06       0
Bank Sta=301.2,320.4
XS Rating Curve= 0 ,0
Exp/Cntr=0.3,0.1

Type RM Length L Ch R = 1 ,10496.9 ,296.3,305.7,315
XS GIS Cut Line= 2
     1591283.202      304790.091     1591957.681      304477.591
#Sta/Elev= 30
       0  820.11    78.2  818.19    97.8  816.18   107.6  814.07   127.2  807.13
   146.7  798.54   156.5  793.52   166.3  785.96   185.8  767.66   195.6  760.89
   205.4  757.68   215.2  755.46   234.7  747.51   244.5  745.03     313  739.14
   336.7  734.81   342.3  733.95   352.1  733.96   361.9  736.01   371.7  739.85
   381.5     742   391.2  742.56   469.5  743.41   518.4  745.94   557.5  749.36
   616.2  757.55     626  759.37   635.8  762.41   645.6   766.6   743.4  810.32
#Mann= 3 , 0 , 0
       0     .06       0   336.7    .045       0   361.9     .06       0
Bank Sta=336.7,361.9
XS Rating Curve= 0 ,0
Exp/Cntr=0.3,0.1

Type RM Length L Ch R = 1 ,10191.2 ,591.7,604.3,616.8
XS GIS Cut Line= 2
     1591349.702       304923.26     1592037.202      304881.594
#Sta/Elev= 30
       0  808.47    68.9  803.06    88.6  800.05   118.1  793.88   127.9  791.28
   137.8  786.92   147.6  779.94   157.4  771.97   167.3  766.04   177.1  763.75
     187  762.77   196.8  760.47   236.2  748.25     246  746.07   255.8  745.04
   265.7  744.58   373.9  740.19   383.7  739.43   393.6  737.64   403.4  735.21
   413.3  734.04   423.1  735.19   432.9   738.5   452.6  746.83     492  761.74
   521.5  774.35   541.2  782.12   590.4  798.61   659.2  822.39   688.8  834.85
#Mann= 3 , 0 , 0
       0     .06       0   403.4    .045       0   432.9      .1       0
Bank Sta=403.4,432.9
XS Rating Curve= 0 ,0
Exp/Cntr=0.3,0.1

Type RM Length L Ch R = 1 ,9586.9  ,710,715.7,721.2
XS GIS Cut Line= 2
     1591162.218      305174.645     1591953.868      305624.649
#Sta/Elev= 30
       0  811.22      49  799.83   137.1  778.21   146.9  776.34   166.5  774.91
   176.2  773.22   264.4  751.49   274.2  749.33     284  747.81   293.8  747.06
   332.9  745.37   489.6  739.55   499.4  738.96   509.2  737.54   522.9  734.68
   528.7   733.8   537.9  733.79   548.3  734.52   567.9  737.39   577.7  738.43
   597.3  739.94   607.1  741.79   616.9  745.95   665.8  773.13   802.9  853.63
   861.6  887.01   871.4  891.64   881.2  895.52     891  898.16   910.6  902.01
#Mann= 3 , 0 , 0
       0     .06       0   522.9    .045       0   537.9      .1       0
Bank Sta=522.9,537.9
XS Rating Curve= 0 ,0
Exp/Cntr=0.3,0.1

Type RM Length L Ch R = 1 ,8871.2  ,312.8,302.8,292.9
XS GIS Cut Line= 2
     1590660.858      305489.729     1591293.619      306096.514
#Sta/Elev= 30
       0  890.02    19.5  880.02      39  871.96    77.9  858.01   175.3  825.84
   204.6   815.3   253.3  795.44   331.2  761.63   340.9  758.89   360.4  755.84
   379.9  748.82   389.6  747.08   399.4  746.28   457.8  743.09   496.8  742.01
   613.7  740.23   623.4  739.43   642.9  734.88   646.9  734.44   652.6  733.82
   661.9  733.77   672.1  734.72   701.4  740.56   711.1  743.33   720.8  747.54
   808.5   793.8   818.2   798.7     828  802.48   837.7  804.45   876.7  808.74
#Mann= 3 , 0 , 0
       0     .08       0   646.9    .045       0   661.9      .1       0
Bank Sta=646.9,661.9
XS Rating Curve= 0 ,0
Exp/Cntr=0.3,0.1

Type RM Length L Ch R = 1 ,8568.4  ,442.6,430.5,418.4
XS GIS Cut Line= 2
     1590426.379      305989.062     1591113.879      306222.395
#Sta/Elev= 30
       0  836.97    19.6  836.69    29.4  835.73    39.2  833.74    49.1  830.61
    68.7  821.66    98.1  807.14   137.4  787.04   176.6  766.34   186.4  761.59
   196.2  758.34     206  757.11   225.6  756.08   343.4  746.71   431.7  740.99
   510.2  734.74   528.1  733.77   539.6   733.7   543.1  733.71   559.2   734.3
   578.8  737.75   598.5  737.18   608.3  738.52   618.1  742.17   627.9  747.56
   667.2   776.9     677  783.62   686.8     788   696.6  789.54     726  790.46
#Mann= 3 , 0 , 0
       0      .1       0   528.1    .045       0   543.1      .1       0
Bank Sta=528.1,543.1
XS Rating Curve= 0 ,0
Exp/Cntr=0.3,0.1

Type RM Length L Ch R = 1 ,8137.9  ,308,292.6,277.2
XS GIS Cut Line= 2
     1590363.549      306551.361     1591071.014       306386.43
#Sta/Elev= 30
       0  891.39    88.4  843.16   117.8  826.93   137.4  815.91   157.1  804.69
   186.5  787.46   206.2  775.73   235.6  757.73   245.4  752.66   255.2  749.85
     265  748.65   274.9  746.92   284.7  743.96   304.3  736.38   314.1  734.01
     324   733.6   333.8  734.65   353.4  738.49   363.2  739.72     373  740.22
   510.5   742.9   618.4  744.64   638.1  745.27   647.9  746.41   657.7  748.62
   667.5  751.58     697  761.25   706.8  764.18   716.6  766.84   726.4  769.12
#Mann= 3 , 0 , 0
       0      .1       0   304.3    .045       0   333.8     .06       0
Bank Sta=304.3,333.8
XS Rating Curve= 0 ,0
Exp/Cntr=0.3,0.1

Type RM Length L Ch R = 1 ,7845.3  ,233.9,233,232.1
XS GIS Cut Line= 2
     1590712.239      306870.386     1591118.757      306349.538
#Sta/Elev= 30
       0  849.88     9.7  844.25    29.2  830.09      68  801.09    87.4  787.22
   126.3  760.34     136  754.09   145.8  750.63   165.2  747.72   174.9  745.01
   184.6  741.47   194.3  737.46     204  734.25   213.8  732.97   223.5  733.61
   233.2  735.15   252.6  737.75   262.3  738.56   310.9  739.53   388.6   740.2
   437.2  741.05   485.8  742.62     515  744.41   524.7  745.56   534.4  747.69
   544.1  750.81     583  764.23   592.7  767.12   612.1  772.01   660.7  783.22
#Mann= 3 , 0 , 0
       0      .1       0   194.3    .045       0   233.2     .06       0
Bank Sta=194.3,233.2
XS Rating Curve= 0 ,0
Exp/Cntr=0.3,0.1
